--- LTLFSHNGCK.prj (project) ---

Proj Title=LTLFSHNGCK
Current Plan=p01
Default Exp/Contr=0,0
English Units
Geom File=g01
Flow File=f01
Plan File=p01
BEGIN DESCRIPTION:
---------- MODELED AS PART OF WVEMD CTP PROGRAM, 2023----------
Stream Name:Little Fishing Creek
Flood Zone:  AFH
Wetzel County, WV
HEC-RAS Version: RAS 6.3
Vertical Datum: NAVD88
Projection: NAD 1983 StatePlane West Virginia S FIPS 4702 (US Feet)
Terrain: 1-meter West Virginia FEMA R3 South Central (collected 2018-2020)
Land Use: 2019 NLCD
Hydrologic Method:
WV SIR2010-5033 regression equations
Additional Model Notes:
Leveraged XS
END DESCRIPTION:
DSS Export Rating Curves= 0
DSS Export Rating Curve Sorted= 0
DSS Export Volume Flow Curves= 0
DXF OffsetX= 0
DXF OffsetY= 0
DXF ScaleX= 0
DXF ScaleY= 0

--- LTLFSHNGCK.p01 (plan) ---

Plan Title=Floodplain
Program Version=6.30
Short Identifier=Floodplain
Geom File=g01
Flow File=f01
Subcritical Flow
K Sum by GR= 0
Std Step Tol= 0.01
Critical Tol= 0.01
Num of Std Step Trials= 20
Max Error Tol= 0.3
Flow Tol Ratio= 0.001
Split Flow NTrial= 30
Split Flow Tol= 0.02
Split Flow Ratio= 0.02
Log Output Level= 0
Friction Slope Method= 1
Unsteady Friction Slope Method= 2
Unsteady Bridges Friction Slope Method= 1
Parabolic Critical Depth
Global Vel Dist= 0 , 0 , 0
Global Log Level= 0
CheckData=True
Encroach Param=-1 ,0,0, 0
Mapping Interval=1HOUR
Computation Time Step Use Courant=        0
Computation Time Step Use Time Series=    0
Computation Time Step Count To Double=0
Computation Time Step Max Doubling=0
Computation Time Step Max Halving=0
Computation Time Step Residence Courant=0
Run HTab= 0
Run UNet= 0
Run Sediment= 0
Run PostProcess= 0
Run WQNet= 0
Run RASMapper= 0
UNET Theta= 0
UNET Theta Warmup= 0
UNET ZTol= 0
UNET ZSATol= 0
UNET MxIter= 0
UNET Max Iter WO Improvement= 0
UNET MaxInSteps= 0
UNET DtIC= 0
UNET DtMin= 0
UNET MaxCRTS= 0
UNET WFStab= 0
UNET SFStab= 0
UNET WFX= 1
UNET SFX= 1
UNET Gravity=32.17405
UNET 1D Methodology=Finite Difference
UNET DSS MLevel= 1
UNET Pardiso=0
UNET DZMax Abort= 0
UNET Use Existing IB Tables= 0
UNET Froude Reduction=False
UNET Froude Limit= 0
UNET Froude Power= 0
UNET D1 Cores= 0
UNET WindReference=Eulerian
UNET WindDragFormulation=Hsu (1988)
UNET D2 Coriolis=0
UNET D2 Cores= 0
UNET D2 Theta= 1
UNET D2 Theta Warmup= 1
UNET D2 Z Tol= 0.01
UNET D2 Volume Tol= 0.01
UNET D2 Max Iterations= 20
UNET D2 Equation= 0
UNET D2 RampUpFraction=0.1
UNET D2 TimeSlices= 1
UNET D2 Turbulence Formulation=Non-Conservative (original)
UNET D2 Eddy Viscosity=0.3
UNET D2 Transverse Eddy Viscosity=0.1
UNET D2 Smagorinsky Mixing=0
UNET D2 BCVolumeCheck=0
UNET D2 Cores=0
UNET D2 SolverType=PARDISO (Direct)
UNET D2 Minimum Iterations= 3
UNET D2 Maximum Iterations= 30
UNET D2 Restart Number= 10
UNET D2 Relaxation Coeff=1.3
UNET D2 SOR Precondition Iterations= 10
UNET D2 ILUT Maximum Fill= 8
UNET D2 ILUT Tolerance=1E-08
UNET D2 Convergence Tolerance=0.00001
UNET D1D2 MaxIter= 0
UNET D1D2 ZTol=0.01
UNET D1D2 QTol=0.1
UNET D1D2 MinQTol=1
Write IC File= 0
Write IC File at Fixed DateTime=0
Write IC File at Sim End=0
Echo Input=False
Echo Parameters=False
Echo Output=False
Write Detailed= 0
HDF Write Warmup=0
HDF Write Time Slices=0
HDF Flush=0
HDF Compression= 1
HDF Chunk Size= 1
HDF Spatial Parts= 1
HDF Use Max Rows=0
HDF Fixed Rows= 1
Calibration Method= 0
Calibration Iterations= 20
Calibration Max Change=0.05
Calibration Tolerance=0.2
Calibration Maximum=1.5
Calibration Minimum=0.5
Calibration Optimization Method= 1
WQ AD Non Conservative
WQ ULTIMATE=-1
WQ Max Comp Step=1HOUR
WQ Output Interval=15MIN
WQ Output Selected Increments= 0
WQ Output face flow=0
WQ Output face velocity=0
WQ Output face area=0
WQ Output face dispersion=0
WQ Output cell volume=0
WQ Output cell surface area=0
WQ Output cell continuity=0
WQ Output cumulative cell continuity=0
WQ Output face conc=0
WQ Output face dconc_dx=0
WQ Output face courant=0
WQ Output face peclet=0
WQ Output face adv mass=0
WQ Output face disp mass=0
WQ Output cell mass=0
WQ Output cell source sink temp=0
WQ Output nsm pathways=0
WQ Output nsm derived pathways=0
WQ Create Restart=0
WQ Fixed Restart=0
WQ System Summary=0
WQ Write To DSS=0
Sorting and Armoring Iterations= 10
XS Update Threshold= 0.02
Bed Roughness Predictor= 0
Hydraulics Update Threshold= 0.02
Energy Slope Method= 1
Volume Change Method= 1
Sediment Retention Method= 0
Sediment TS Multiplier= 1
Warm Up Method= 0
XS Weighting Method= 0
Number of US Weighted Cross Sections= 1
Number of DS Weighted Cross Sections= 1
Upstream XS Weight=0
Main XS Weight=1
Downstream XS Weight=0
Number of DS XS's Weighted with US Boundary= 1
Upstream Boundary Weight= 1
Weight of XSs Associated with US Boundary= 0
Number of US XS's Weighted with DS Boundary= 1
Downstream Boundary Weight= 0.5
Weight of XSs Associated with DS Boundary= 0.5
Percentile Method= 0
Sediment Output Level= 3
Mass or Volume Output= 0
Output Increment Type= 1
Profile and TS Output Increment= 1
Transport Output Increment 1
XS Output Flag= 0
XS Output Increment= 10
Read HDF5 Sediment Hotstart= 0
Sediment Hotstart Type= 0
Write Gradation File= 0
Read Gradation Hotstart= 0
Write HDF5 File= 1
Write Binary Output= 1
Write DSS Sediment File= 0
DSS Sediment Output Type= 1
SV Curve= 0
Specific Gage Flag= 0
Subcell Erosion Methods= 0
Subcell Deposition Methods= 0
Advection Scheme= 1
Matrix Solver= 0
Implicit Weighting Factor= 1
Maximum Outer Loop Convergence Iterations= 5
Convergence Maximum Absolute= 0.001
Convergence RMSE= 0.0001
Grain Fractions Max Abs Error= 0.001
Max Subgrid Regions= 1
Max Subgrid Length Scale= 3.402823E+38
Initial Layer Thickness= 3.402823E+38
Min Layer Thickness= 3.402823E+38
Max Layer Thickness= 3.402823E+38
Number of Layers= 5

--- LTLFSHNGCK.f01 (steady flow) ---

Flow Title=Flow
Program Version=6.30
Number of Profiles= 1
Profile Names=F01pct
River Rch & RM=River 1,Reach 1,106220
     629
River Rch & RM=River 1,Reach 1,104016
     733
River Rch & RM=River 1,Reach 1,102744
     921
River Rch & RM=River 1,Reach 1,100011
    1030
River Rch & RM=River 1,Reach 1,97965
    1160
River Rch & RM=River 1,Reach 1,93630
    1590
River Rch & RM=River 1,Reach 1,88506
    1810
River Rch & RM=River 1,Reach 1,84506
    2510
River Rch & RM=River 1,Reach 1,80006
    2790
River Rch & RM=River 1,Reach 1,77001
    3840
River Rch & RM=River 1,Reach 1,65506
    4930
River Rch & RM=River 1,Reach 1,58506
    5480
River Rch & RM=River 1,Reach 1,47500
    6120
River Rch & RM=River 1,Reach 1,31500
    6800
Boundary for River Rch & Prof#=River 1,Reach 1         , 1
Up Type= 0
Dn Type= 3
Dn Slope=0.00153
DSS Import GetInterval= 0
DSS Import GetPeak= 0
DSS Import FillOption= 0

--- LTLFSHNGCK.g01 (geometry) ---

Geom Title=Geometry
Program Version=6.30

River Reach=River 1         ,Reach 1
Reach XY= 30
1660456.90894088412091.0222445581658214.08632681412427.365403891
1652490.69816731 409544.593938471644790.97340931409233.330453396
1641223.42608248413149.5152063071635842.30856389414319.302892983
1631555.16950038410949.9753140661627097.49468872412157.506363556
1624926.57777072411647.9532488141624702.96076389410072.370441973
1622014.19678447409333.5182451461620883.06469797407148.838715299
1617403.24340796410409.2162249831616430.64758414407935.912444562
1614369.75177155406765.1313215641612709.80856913408321.972367972
1612422.26846181406225.563831151 1609826.3878268406327.520320147
1610453.01911947404755.7869150641608977.51419647403323.813729137
1605602.64004073 404871.490095721606859.33962706406060.600578398
1605899.34482789 407109.95051381 1603256.4954548405758.167784303
1602185.37981489407513.1941298991599833.50722206404635.501066387
1597986.83473431408945.1669877321597434.66589114407162.646930724
1595559.35402498409107.8392345611593461.39463823408542.023108974

Type RM Length L Ch R = 1 ,106220  ,216.8,217.3,217.4
BEGIN DESCRIPTION:
Structure 26 XS 4
END DESCRIPTION:
XS GIS Cut Line= 3
1660446.24087117411623.6280793461660347.69587546411970.234615963
1660419.05604476412637.961914447
#Sta/Elev= 30
       0 1174.92    42.5  1165.5    92.4 1147.48   129.9 1138.38   179.8 1114.19
   208.9 1107.12   277.7 1071.26   308.7 1062.11   362.8  1036.9   463.2 1033.22
   475.3 1029.46   479.3 1028.75   484.1 1029.32   503.5 1032.43   527.6 1033.03
   539.7 1038.16   571.8  1035.4   575.9 1036.53   579.9 1040.45   588.1 1054.63
     608 1066.75   692.5 1096.43   772.3 1131.29   805.2  1142.2   821.3 1143.45
   865.5 1157.75   929.8 1180.06   970.1 1196.14     993 1202.51  1031.9 1209.72
#Mann= 6, -1 ,  0
       0     0.1       0  420.34    0.05       0   475.3   0.045       0
   484.1    0.05       0  510.34    0.06       0  610.34     0.1       0
Bank Sta=475.3,484.1
XS Rating Curve= 0 ,0
Exp/Cntr(USF)=0,0
Exp/Cntr=0.3,0.1

Type RM Length L Ch R = 1 ,106002  ,24.8,24.7,24.6
BEGIN DESCRIPTION:
Structure 26 XS 3
END DESCRIPTION:
XS GIS Cut Line= 4
1660412.54267352411610.330663648 1660137.2963062411923.805693089
1660155.64606402412206.6977928281660216.81192343412744.957355575
#Sta/Elev= 30
       0 1176.88    61.4 1164.32    98.2 1150.58   146.7 1140.71   182.5 1120.42
   231.5 1103.85   288.1 1075.58   396.8  1041.5   598.3 1030.64  609.65 1025.75
   614.3 1024.66  620.711025.663   642.4 1033.56   666.4  1034.8   698.5 1031.68
   702.5 1034.56   714.6 1051.38     783 1077.87   797.6 1081.03   831.3 1099.49
   883.9 1121.52     916 1133.71   964.2 1146.43   984.3 1155.65   999.2  1157.5
  1044.7 1171.83    1089 1191.41  1153.4 1211.08  1226.9 1241.83  1242.4 1245.32
#Mann= 6, -1 ,  0
       0     0.1       0  417.17    0.06       0  517.17    0.05       0
  609.65   0.045       0  620.71    0.06       0  720.65     0.1       0
Bank Sta=609.65,620.71
XS Rating Curve= 0 ,0
Exp/Cntr(USF)=0,0
Exp/Cntr=0.3,0.1

Type RM Length L Ch R = 1 ,105978  ,21.2,21.2,21.3
BEGIN DESCRIPTION:
Structure 26 XS 2
END DESCRIPTION:
XS GIS Cut Line= 4
1660400.30950163411584.3351734021660109.77166947411922.276546604
1660132.70886675412214.343525254 1660198.4621656412758.719673941
#Sta/Elev= 30
       0 1180.65    71.2 1164.53   153.5 1141.29   184.4 1127.27   202.8 1115.14
   235.7 1105.46   298.1 1074.43   338.5 1059.76   399.1 1043.11   632.5 1030.98
   644.5 1025.34   648.5 1024.25   654.6 1025.29   654.6  1025.3   672.6 1033.02
   732.8 1031.57   748.9 1049.93   801.2 1071.32   813.4 1072.06   865.7 1098.66
   914.1 1117.93   998.7 1145.48  1022.9 1158.42  1063.2 1164.56    1096 1176.17
  1123.6 1190.51  1188.1 1210.58  1239.8 1229.93  1257.7 1240.04    1287 1248.15
#Mann= 6, -1 ,  0
       0     0.1       0  445.66    0.06       0  545.66    0.05       0
   644.5   0.045       0   654.6    0.06       0  748.63     0.1       0
Bank Sta=644.5,654.6
XS Rating Curve= 0 ,0
Exp/Cntr(USF)=0,0
Exp/Cntr=0.3,0.1

Type RM Length L Ch R = 1 ,105957  ,38.5,38.7,39.2
BEGIN DESCRIPTION:
Structure 25 XS 3
END DESCRIPTION:
XS GIS Cut Line= 4
1659507.33135917411638.571795728 1660088.4070235411932.167920862
1660111.34422078412207.4142881761660177.09751964412759.436169289
#Sta/Elev= 30
       0 1281.37    45.7 1270.37   144.3 1234.62   278.9  1176.2   395.3  1136.4
   475.9 1102.47   517.1 1082.47   616.4 1046.41   671.5 1038.97     828 1031.57
  842.531025.292   848.1 1023.69  854.451025.361   868.2  1032.6   900.3 1034.29
   932.4 1031.62   944.5 1046.37   952.5 1051.68   988.8 1066.06  1004.9 1066.68
  1033.3 1082.84  1097.6 1106.62  1137.8 1125.41  1198.3 1145.01  1234.5  1160.9
  1281.7  1168.2  1327.2 1189.71  1427.9 1223.99  1460.1 1240.52  1483.2 1247.41
#Mann= 7, -1 ,  0
       0     0.1       0     640    0.06       0  741.04    0.05       0
  841.04    0.06       0  842.53   0.045       0  854.45    0.06       0
  937.24     0.1       0
Bank Sta=842.53,854.45
XS Rating Curve= 0 ,0
Exp/Cntr(USF)=0,0
Exp/Cntr=0.3,0.1

Type RM Length L Ch R = 1 ,105918  ,141.6,145.7,152.8
BEGIN DESCRIPTION:
Structure 25 XS 2
END DESCRIPTION:
XS GIS Cut Line= 4
1659523.25250973 411659.359506961660053.86634005 411960.60136452
1660070.68695138412189.9733372821660176.19805885 412767.99070864
#Sta/Elev= 30
       0 1278.21   111.4 1238.99   263.2 1174.36   375.1 1135.31   462.1  1099.5
   512.8 1075.68   579.5 1051.28     603  1039.4   758.5 1030.66   766.5 1029.23
   774.5 1023.69   782.6 1022.31   794.6 1023.76   802.6 1027.66   826.7 1029.45
   840.1 1033.55   871.2 1031.78   895.6 1053.69   915.9 1061.34   940.3 1063.66
   952.5 1070.39   993.2 1083.58  1086.7 1130.25  1123.3 1139.92    1168  1157.7
  1233.1 1171.61  1265.6 1189.13  1363.2 1223.36  1395.7 1240.14  1427.7 1250.74
#Mann= 6, -1 ,  0
       0     0.1       0  770.16    0.05       0   774.5   0.045       0
   794.6    0.05       0  850.15    0.06       0  870.15     0.1       0
Bank Sta=774.5,794.6
XS Rating Curve= 0 ,0
Exp/Cntr(USF)=0,0
Exp/Cntr=0.3,0.1

Type RM Length L Ch R = 1 ,105772  ,268.5,260.8,248.7
BEGIN DESCRIPTION:
Structure 25 XS 1
END DESCRIPTION:
XS GIS Cut Line= 6
1659446.36331833411658.9633951391659943.76117658412108.403628957
1659928.71208145412128.4690891351659914.66625933412165.590190462
 1659897.6130818412250.6235628731660098.10117651 412809.61155575
#Sta/Elev= 30
       0 1292.55    84.5 1271.76   115.7 1256.89   174.9 1236.38   226.1 1211.81
   266.5 1197.99   395.9 1138.96   427.2 1130.59   521.4 1076.75   622.3 1030.51
   636.7 1026.64   680.5 1025.43   704.1 1021.46   712.6 1020.64   730.1 1021.48
   831.7 1031.84     858 1030.05   862.3 1032.63   870.8 1047.61   883.5 1055.67
   934.5 1070.81   985.5 1095.34  1016.3 1103.77  1070.5  1128.9  1125.8  1139.8
  1202.2 1164.87    1232 1183.57  1244.6 1185.42  1270.2 1199.52  1415.9 1258.52
#Mann= 6, -1 ,  0
       0     0.1       0   704.1   0.045       0   730.1     0.1       0
  796.98    0.07       0  892.01    0.06       0 1002.01     0.1       0
Bank Sta=704.1,730.1
XS Rating Curve= 0 ,0
Exp/Cntr(USF)=0,0
Exp/Cntr=0.3,0.1

Type RM Length L Ch R = 1 ,105511  ,499.4,500.5,501.4
XS GIS Cut Line= 6
1659373.76740642411701.4954645931659618.85418659412110.830603927
1659707.90748617412261.7046460061659921.84964359412659.323929504
1659960.94864675 412750.917578341659996.77337825412844.759254172
#Sta/Elev= 30
       0 1296.11      36 1283.57    78.1 1273.22   121.5 1249.91   183.7 1227.32
   283.3 1174.43   336.4 1155.58   394.7 1128.27   432.5 1105.75   520.9 1071.13
   540.6 1060.36   567.4 1035.42593.20061018.189   601.9 1017.38609.55051018.198
   720.3  1024.6     749 1031.27   778.6 1028.61   796.2 1043.02     819 1055.76
     869 1074.92   982.3 1128.48  1014.3 1137.12  1055.2 1155.89    1087 1163.15
  1148.6 1192.96  1161.7 1194.54  1222.3 1221.97    1248 1236.68  1303.9 1254.64
#Mann= 6, -1 ,  0
       0     0.1       0593.2006   0.045       0609.5505    0.06       0
  722.29    0.07       0  797.34    0.06       0  834.85     0.1       0
Bank Sta=593.2006,609.5505
XS Rating Curve= 0 ,0
Exp/Cntr(USF)=0,0
Exp/Cntr=0.3,0.1

Type RM Length L Ch R = 1 ,105011  ,497.2,499.6,502.9
XS GIS Cut Line= 6
1659021.08602518411796.7272295061659053.45374259411893.194884345
1659117.70787917 412080.115770341659208.12174034412343.134273171
1659444.05926059413029.4957613351659476.43977326413123.695048004
#Sta/Elev= 30
       0  1365.8    33.6 1353.98   113.7 1310.06   147.6 1285.97   181.4 1269.24
   200.9 1264.24   236.4 1242.24   278.7 1226.62   323.7 1204.14   346.4 1187.45
   367.5 1183.39   401.4 1161.33   439.4 1150.23   473.3 1129.04   515.6 1115.31
   549.4 1093.37     651 1046.11   685.7 1016.19  697.621009.644   701.7 1009.16
   707.7 1009.63   828.6 1014.73   849.7 1023.71   883.6 1025.67   921.7 1055.64
  1022.5 1096.94  1065.4 1119.04  1166.3 1153.12  1302.6 1186.15  1402.9  1193.3
#Mann= 6, -1 ,  0
       0     0.1       0  652.53    0.05       0  697.62   0.045       0
   707.7    0.05       0  812.53    0.06       0  965.03     0.1       0
Bank Sta=697.62,707.7
XS Rating Curve= 0 ,0
Exp/Cntr(USF)=0,0
Exp/Cntr=0.3,0.1

Type RM Length L Ch R = 1 ,104511  ,507.3,495.6,484.6
XS GIS Cut Line= 6
1658887.42192243411787.6632712481658767.98449726412426.993029341
1658750.48650075412525.4541185051658728.32873668 412686.62604025
1658691.08766942412973.7320933341658686.03309368 413037.63830109
#Sta/Elev= 30
       0    1325     107 1274.46   144.2 1265.47   188.7 1243.02   261.3 1224.69
   363.6 1187.47   407.8 1159.24   440.4 1149.48   481.1 1123.69   497.4 1120.99
   517.7 1112.89   542.1 1096.41   599.1 1064.43   627.5 1053.66     656 1038.63
   676.3 1023.34   688.5 1007.08   696.6 1002.92   704.8 1001.94   710.3  1002.9
   785.8 1007.67     806  1012.6   846.4 1013.75   850.4 1018.26   858.5 1034.34
   862.5 1037.88   898.9 1054.16  1000.6 1072.14  1132.7 1117.88  1266.7 1153.92
#Mann= 7, -1 ,  0
       0     0.1       0   696.6   0.045       0   710.3     0.1       0
  740.39    0.05       0  845.47    0.06       0  943.08    0.05       0
 1242.59     0.1       0
Bank Sta=696.6,710.3
XS Rating Curve= 0 ,0
Exp/Cntr(USF)=0,0
Exp/Cntr=0.3,0.1

Type RM Length L Ch R = 1 ,104016  ,41.8,53.4,65.1
BEGIN DESCRIPTION:
Structure 24 XS 4
END DESCRIPTION:
XS GIS Cut Line= 6
1658522.62097305411786.1664462451658248.90375223412406.999919186
1658288.66156084412446.0263417741658305.48343938412460.654062244
1658367.65125137412473.8190106661658621.54203438413025.395975623
#Sta/Elev= 30
       0 1217.32    68.2 1192.07   125.1 1177.41   146.9    1169   168.7 1157.96
   237.3 1144.99   264.6 1137.83   307.1 1120.53   353.2 1111.37   426.6 1079.15
   495.2  1046.6   580.1 1023.45   614.6 1016.96   636.5 1009.06  696.82995.6078
   715.4  995.12  723.19995.6077   820.1 1001.07   862.7 1006.23   946.4 1006.82
   993.4 1020.75  1018.5 1026.05  1063.7 1043.43  1105.9  1053.2  1126.9 1054.71
  1140.1 1060.88  1271.8 1095.07  1318.6 1112.07  1353.2 1118.11  1427.3 1138.31
#Mann= 10, -1 ,  0
       0     0.1       0  696.82   0.045       0  723.19    0.06       0
  754.24    0.07       0  870.08    0.06       0  980.08     0.1       0
 1130.08    0.05       0 1190.08     0.1       0 1370.08    0.05       0
 1410.08     0.1       0
Bank Sta=696.82,723.19
XS Rating Curve= 0 ,0
Exp/Cntr(USF)=0,0
Exp/Cntr=0.3,0.1

Type RM Length L Ch R = 1 ,103962  ,63.3,63.2,63.1
BEGIN DESCRIPTION:
Structure 24 XS 3
END DESCRIPTION:
XS GIS Cut Line= 3
1658503.42168941411764.7583954541658180.60187589412520.836379741
1657738.84844687412836.859986657
#Sta/Elev= 30
       0 1213.99    25.9 1199.58    34.6  1200.3    47.6 1197.19     173 1153.66
     239 1141.99   304.2 1118.83   352.1 1106.29   504.3 1044.07     613 1017.39
   670.6 1007.99   691.2 1000.73   706.4 1000.72   717.4  993.03   721.8  992.34
  729.23993.0525   741.9 1000.99   756.5 1002.64     800  998.06   857.1  1001.5
   879.6 1015.39   921.1 1048.15   955.5  1060.7  1048.9 1104.75    1076 1114.65
  1127.6 1138.61  1176.8 1154.66  1192.8 1163.67  1265.3 1185.22  1365.3 1224.51
#Mann= 5, -1 ,  0
       0     0.1       0     710    0.06       0   717.4   0.045       0
  729.23    0.06       0     820     0.1       0
Bank Sta=717.4,729.23
XS Rating Curve= 0 ,0
Exp/Cntr(USF)=0,0
Exp/Cntr=0.3,0.1

Type RM Length L Ch R = 1 ,103899  ,386.6,388,390.4
BEGIN DESCRIPTION:
Structure 24 XS 2
END DESCRIPTION:
XS GIS Cut Line= 3
1658440.55677836411734.1754657521658124.53317144 412493.65155334
1657699.77025892412818.170418506
#Sta/Elev= 30
       0 1206.46    15.6 1201.34    32.9 1190.06    97.9 1170.64   145.5  1147.7
   175.9 1139.12   204.1 1122.87   232.2 1114.75   258.2 1100.89   286.7 1101.84
   320.3 1089.84   396.8 1087.69   500.8 1060.25   557.1 1034.36   630.8 1013.89
   661.1 1001.87   705.8  998.65  722.87992.1537   730.3  991.03   734.7  992.24
   745.6  999.59   765.1 1001.93   828.2  998.01   878.5 1036.25   965.7  1071.4
  1101.8 1134.38  1163.4 1152.38  1196.3  1170.6  1290.1 1200.13  1357.1 1227.09
#Mann= 5, -1 ,  0
       0     0.1       0  722.87   0.045       0   734.7     0.1       0
     740    0.06       0   862.6     0.1       0
Bank Sta=722.87,734.7
XS Rating Curve= 0 ,0
Exp/Cntr(USF)=0,0
Exp/Cntr=0.3,0.1

Type RM Length L Ch R = 1 ,103511  ,502.2,500.2,496.8
BEGIN DESCRIPTION:
Structure 24 XS 1
END DESCRIPTION:
XS GIS Cut Line= 6
1658310.92241925411635.8555040061657823.97457425412206.791698083
1657778.22499384412266.3480094221657668.79017334412411.469766423
1657549.01219767412566.6964900941657423.92550559412721.898935586
#Sta/Elev= 30
       0 1233.82    59.8 1211.15    90.6 1206.21   142.9 1190.09   189.7    1182
   279.6 1175.56     327 1156.17   371.3 1145.99   405.9 1130.08   421.6 1118.59
     469  1103.2   552.6    1052   577.3 1043.41   651.2 1003.78  691.45988.1398
   700.2  985.74   710.7  988.03   762.7  989.29   782.9  994.28   833.2  992.05
   877.1 1024.78   902.4 1039.53  1003.6 1089.88  1048.9 1107.39  1094.3 1131.34
  1210.8 1177.78  1292.7  1198.7  1336.2 1205.63  1370.6 1206.23  1402.7 1200.47
#Mann= 5, -1 ,  0
       0     0.1       0  691.45   0.045       0   710.7     0.1       0
  770.39    0.06       0  895.49     0.1       0
Bank Sta=691.45,710.7
XS Rating Curve= 0 ,0
Exp/Cntr(USF)=0,0
Exp/Cntr=0.3,0.1

Type RM Length L Ch R = 1 ,103011  ,267.1,266.7,263.5
BEGIN DESCRIPTION:
Structure 23 XS 4
END DESCRIPTION:
XS GIS Cut Line= 6
1657719.63160709  411283.59439751657559.18835843411643.630422845
1657342.99292468412115.1826293321657305.40113634412201.082720011
1657280.31522851412295.8135016711657222.21232635412594.335214332
#Sta/Elev= 30
       0    1196    31.7  1189.7    54.9 1180.39   101.7 1173.47   171.7 1153.19
   303.9 1136.48   457.6 1100.97   498.4 1079.97   526.9 1070.13   572.3 1044.69
   613.3 1027.54   637.1  1020.3   694.3  980.91   703.1  979.38  713.02981.0554
   779.5  983.74   804.5  988.75   830.8  988.56   848.4 1000.33   874.8 1006.54
   883.6 1012.89   949.3 1037.36  1039.2 1056.44  1068.2 1060.15  1088.9 1056.63
  1121.8 1063.08  1195.3  1069.2  1264.5 1069.53    1350  1077.2  1408.8 1084.93
#Mann= 6, -1 ,  0
       0     0.1       0   694.3   0.045       0  713.02    0.06       0
  750.42    0.07       0  810.42    0.06       0  922.92     0.1       0
Bank Sta=694.3,713.02
XS Rating Curve= 0 ,0
Exp/Cntr(USF)=0,0
Exp/Cntr=0.3,0.1

Type RM Length L Ch R = 1 ,102744  ,48.7,48.3,46.4
BEGIN DESCRIPTION:
Structure 23 XS 3
END DESCRIPTION:
XS GIS Cut Line= 5
1657423.59505552411200.084125758 1657216.6101434411807.127121968
1657175.07464083411923.6071182961657126.68134444 412076.31995005
 1656782.6233853412293.458750931
#Sta/Elev= 30
       0 1162.94    50.4 1143.85    85.2 1133.65   109.9 1113.63   135.5 1112.52
   221.5 1096.12   317.4 1062.31   356.1 1055.92     457 1025.59   516.1 1001.28
   583.7  991.75   604.8  984.46   714.9  979.37   730.5  975.66   736.3  975.22
     743  975.81   761.9  986.54   806.4  984.93     933   989.1   956.6 1003.28
   999.2 1020.09  1017.1 1030.94  1084.3 1063.45  1098.5  1064.9  1130.2 1084.88
  1155.3 1097.32  1174.2 1100.02  1237.5 1132.31  1306.7 1160.95  1332.1 1166.59
#Mann= 6, -1 ,  0
       0     0.1       0  661.36    0.05       0   730.5   0.045       0
     743    0.05       0  765.03    0.06       0  875.03     0.1       0
Bank Sta=730.5,743
XS Rating Curve= 0 ,0
Exp/Cntr(USF)=0,0
Exp/Cntr=0.3,0.1

Type RM Length L Ch R = 1 ,102696  ,184.6,185.6,189.6
BEGIN DESCRIPTION:
Structure 23 XS 2
END DESCRIPTION:
XS GIS Cut Line= 4
1657386.96038006411180.9886578241657173.00572783411730.558450814
1657114.54539713412006.4550735291656766.42049456412269.324897912
#Sta/Elev= 30
       0 1175.67    29.9 1166.49    63.6 1147.03    98.2 1139.11   136.9 1136.38
   196.5 1123.94   231.3 1113.65   308.6 1099.48   428.8 1060.79   497.4 1035.06
     558 1007.55   591.8  989.42   624.5  983.98   714.4   980.2   730.5  975.54
     739  975.17  745.19975.6585   767.7  986.14   845.3  985.22   871.8  991.77
   895.1 1006.11   970.1 1037.49   988.1 1042.89  1045.2 1073.27  1060.3 1074.82
  1090.3 1092.19  1110.4  1099.6  1125.4 1101.43  1200.5 1139.95    1308 1173.85
#Mann= 6, -1 ,  0
       0     0.1       0  689.75    0.05       0   730.5   0.045       0
  745.19    0.05       0  789.75    0.06       0  901.77     0.1       0
Bank Sta=730.5,745.19
XS Rating Curve= 0 ,0
Exp/Cntr(USF)=0,0
Exp/Cntr=0.3,0.1

Type RM Length L Ch R = 1 ,102510  ,500.8,499.8,497.7
BEGIN DESCRIPTION:
Structure 23 XS 1
END DESCRIPTION:
XS GIS Cut Line= 6
1657362.43579917411168.8866216691657278.72402434411351.421361595
 1657225.8980145411434.6167332531657020.14088009411721.750345334
1656828.99920201412024.6024299261656608.08527376412355.724471092
#Sta/Elev= 30
       0  1182.8    21.4 1177.74    95.4 1150.32   130.9 1148.59   179.9 1140.92
   254.3 1133.95   402.4 1100.67   422.5 1091.69   445.4 1076.97   511.3 1040.38
   568.7 1015.32   585.9 1003.67   616.7  977.12   683.7  975.52   695.2  972.94
   703.4   972.2  710.04972.8776   722.4  975.87   764.3  978.18   779.3  984.53
   811.2  984.51     836 1007.33   857.6 1021.31   892.5 1037.11  1001.2  1093.5
    1049 1110.66  1092.7 1133.58  1144.8 1156.62  1318.3 1212.79  1408.9 1232.32
#Mann= 6, -1 ,  0
       0     0.1       0  662.67    0.05       0   695.2   0.045       0
  710.04    0.05       0  782.67    0.06       0  898.06     0.1       0
Bank Sta=695.2,710.04
XS Rating Curve= 0 ,0
Exp/Cntr(USF)=0,0
Exp/Cntr=0.3,0.1

Type RM Length L Ch R = 1 ,102011  ,501.7,499.7,496.8
XS GIS Cut Line= 6
1656777.06754734410903.4964044241656722.85735393411099.935316011
1656698.54998784411196.2136667521656667.96835609411288.282052174
1656537.08804043411619.6196440911656285.61413392412219.606633082
#Sta/Elev= 30
       0 1269.18    88.4 1238.56   109.1 1224.09     134 1213.69   154.7  1211.4
   245.7 1171.28   278.7 1162.84   316.1 1144.87   345.6 1136.25   379.3 1121.39
   409.4 1104.21   447.6  1092.7   483.5 1067.64   589.5 1020.45   606.7 1015.16
   671.2   974.3     697  967.96   705.9  966.22  719.58968.1961   770.3  970.47
   791.5  976.59     831  976.06   891.7 1019.31  1018.1 1089.74  1054.4 1104.02
  1112.9 1132.58  1208.3 1166.08  1282.1 1196.97  1325.5 1207.94  1406.9 1238.21
#Mann= 6, -1 ,  0
       0     0.1       0     697   0.045       0  719.58     0.1       0
  766.35    0.07       0  786.35    0.06       0  871.37     0.1       0
Bank Sta=697,719.58
XS Rating Curve= 0 ,0
Exp/Cntr(USF)=0,0
Exp/Cntr=0.3,0.1

Type RM Length L Ch R = 1 ,101511  ,495.2,500,504.5
XS GIS Cut Line= 6
 1656218.5224046410761.3857962491656195.81050776410858.790785179
1656174.33548509410955.9411814211656132.94842875411147.096310928
1656114.32215367411239.0206677621655960.08000809 412138.78658475
#Sta/Elev= 30
       0 1271.22    19.7 1260.24    81.3 1242.78   134.6 1219.88   183.7 1203.24
   253.3 1169.01   292.8 1154.93   396.6 1102.03   449.6 1084.55   461.9 1079.08
   486.4 1061.79   514.8 1051.66   539.1  1038.3   608.1 1011.96   644.6  990.63
   677.1  965.75   689.3  962.38   701.5  961.56  712.94962.4349   731.2  968.45
   754.2  968.98   774.5  965.56   871.9   970.6   940.9 1016.75   985.5 1040.91
  1054.5 1084.45  1091.1  1099.4  1143.4 1127.99  1212.9 1150.09  1401.8 1180.26
#Mann= 4, -1 ,  0
       0     0.1       0   689.3   0.045       0  712.94    0.06       0
  886.39     0.1       0
#XS Ineff= 2 , 0
                          756.87         1009.74
Permanent Ineff=
       F       F
Bank Sta=689.3,712.94
XS Rating Curve= 0 ,0
Exp/Cntr(USF)=0,0
Exp/Cntr=0.3,0.1

Type RM Length L Ch R = 1 ,101011  ,494,499.3,504.5
XS GIS Cut Line= 6
1656051.57916893410688.0640925021655854.73343401410918.464222252
1655793.94976293410995.2869032621655690.14813326411144.267576426
1655648.33095968411206.6086590891655257.03974751411846.903310254
#Sta/Elev= 30
       0 1283.94    59.5  1254.6   130.5 1228.75   195.7 1198.97   221.2 1182.01
   258.6  1165.2   300.7 1152.03   351.9 1121.95   378.2 1113.04   407.4 1095.46
   440.6 1085.74     537 1034.64     607  1007.2   669.3  967.63  694.47957.3945
   706.8  953.99   720.9  957.29   730.2  963.16   752.3  964.94   778.5  958.24
   842.2  957.92   877.4  962.65   895.9  972.49   912.3  989.94   941.4 1009.63
  1060.7 1076.94  1100.6 1089.48  1177.1 1130.24  1337.8 1176.82    1408 1187.59
#Mann= 5, -1 ,  0
       0     0.1       0  677.65    0.06       0  694.47   0.045       0
   720.9    0.06       0  807.65     0.1       0
#XS Ineff= 2 , 0
                          749.96          992.24
Permanent Ineff=
       F       F
Bank Sta=694.47,720.9
XS Rating Curve= 0 ,0
Exp/Cntr(USF)=0,0
Exp/Cntr=0.3,0.1

Type RM Length L Ch R = 1 ,100512  ,506.5,500.7,491.4
XS GIS Cut Line= 6
1655899.53583784410484.1327418391655353.01462117410836.726524845
1655269.70835733410892.0604036751655057.61855842411039.614898592
1654976.94385101411094.7798145121654728.56770734411261.418588832
#Sta/Elev= 30
       0 1179.01    81.9 1177.91   137.4 1168.81   246.8 1162.16     318 1149.17
     376 1119.68   408.7 1111.17     442 1093.22   470.6 1084.91   503.3 1064.73
   532.5 1051.92   584.8 1022.24   613.4 1012.56   661.1  981.67   685.1  960.99
   693.4  950.22     700  948.81   709.1  950.38   718.7  953.19   829.5  952.59
   852.5  958.69   891.3  955.55   905.3  963.08   942.4  995.43  1059.4 1057.37
  1085.3 1074.39  1122.8 1085.55    1212 1134.63  1252.3 1149.12  1405.6 1216.74
#Mann= 6, -1 ,  0
       0     0.1       0   693.4   0.045       0   709.1     0.1       0
   780.4    0.05       0   835.8    0.06       0 1004.09     0.1       0
Bank Sta=693.4,709.1
XS Rating Curve= 0 ,0
Exp/Cntr(USF)=0,0
Exp/Cntr=0.3,0.1

Type RM Length L Ch R = 1 ,100011  ,494.6,500,504.8
XS GIS Cut Line= 6
1655133.97175217409824.235439584  1654957.002946410630.431005672
1654931.35043825   410714.3888431654895.31343684410803.790895179
1654844.00054733410894.2575777621654658.81751876 411158.42732501
#Sta/Elev= 30
       0 1332.12    38.8 1321.05   155.9 1256.21   217.4 1230.73   250.1 1208.51
   299.3 1186.71   344.3 1152.91   377.1 1140.02   454.9 1090.13     504 1074.65
   564.6 1032.39   614.6 1007.27   663.7  976.63   692.4  946.07   700.3  943.59
  712.44945.9859   902.9  948.92   938.8  956.16   971.6  955.92   993.1  976.47
  1028.8  1003.1    1080 1027.79  1145.1 1066.95  1178.7 1076.12  1213.3 1095.86
  1233.4 1102.82  1280.7 1132.82  1336.7 1156.49  1364.5 1174.98  1436.3 1204.23
#Mann= 5, -1 ,  0
       0     0.1       0   692.4   0.045       0  712.44     0.1       0
  845.39    0.06       0 1059.57     0.1       0
Bank Sta=692.4,712.44
XS Rating Curve= 0 ,0
Exp/Cntr(USF)=0,0
Exp/Cntr=0.3,0.1

Type RM Length L Ch R = 1 ,99511   ,503.2,500,496.9
XS GIS Cut Line= 6
1654919.98760009409773.2184812581654868.87680992409860.298687667
1654758.19724126410024.9755236661654215.38172585410748.723420009
1654163.45236775410833.7606514991654116.58435126410922.801155835
#Sta/Elev= 30
       0 1241.39    17.8 1232.92   109.7 1202.65   161.3  1194.8   185.6 1185.27
   251.8 1146.21   296.1 1131.81   333.9 1107.08   368.9 1095.62   383.9 1084.11
   438.9 1067.72   474.9 1044.14   533.9 1018.31   556.2 1004.32   578.9  998.11
   643.9  966.14   668.9  946.92   688.9  940.93   698.9  938.56   713.9  941.06
   863.9  942.21   888.9  946.74   918.9  946.42   996.2  994.64  1083.9 1029.03
  1113.9 1037.78  1163.9 1060.66  1236.7 1082.72  1292.9 1090.26  1404.4 1091.76
#Mann= 6, -1 ,  0
       0     0.1       0   688.9   0.045       0   713.9     0.1       0
  802.54    0.05       0  827.54    0.06       0  955.04     0.1       0
Bank Sta=688.9,713.9
XS Rating Curve= 0 ,0
Exp/Cntr(USF)=0,0
Exp/Cntr=0.3,0.1

Type RM Length L Ch R = 1 ,99011   ,497.4,500,500.8
XS GIS Cut Line= 6
1654332.80701593409519.9729247541654291.68078583409610.738491252
1654252.42331843409701.8652774991654214.31873584409792.628547415
1654106.65294068410049.0686513331653787.13750359410810.107155502
#Sta/Elev= 30
       0 1247.18    18.2 1238.67   110.3 1214.15   207.3 1162.61   240.8 1150.55
   263.1 1136.46   295.9 1125.15   315.4 1114.07   388.3 1090.03     423 1070.55
   453.4 1063.11   483.8 1040.55   518.5 1024.83   557.5 1002.29   622.6     979
   653.4  963.75   687.7  934.35   702.2  933.63   710.6934.3844   813.5  938.22
   839.7  945.28   902.3  942.52    1000  948.38    1047   946.9  1147.5   961.1
  1181.3  971.28  1238.6  981.32  1264.6  978.15    1353  985.72  1400.8   984.4
#Mann= 8, -1 ,  0
       0     0.1       0   687.7   0.045       0   710.6    0.05       0
  800.43    0.06       0 1006.68    0.05       0 1113.56    0.06       0
 1193.56    0.05       0    1222     0.1       0
Bank Sta=687.7,710.6
XS Rating Curve= 0 ,0
Exp/Cntr(USF)=0,0
Exp/Cntr=0.3,0.1

Type RM Length L Ch R = 1 ,98511   ,548.2,546.1,543.5
BEGIN DESCRIPTION:
Structure 22 XS 4
END DESCRIPTION:
XS GIS Cut Line= 6
1654010.05241209409343.7255738381653599.09621301 409971.58028926
1653438.26385751 410176.52476126 1653386.0359436410262.920257762
1653336.88151434410353.0040670931653243.07395917410536.274041757
#Sta/Elev= 30
       0 1203.35   114.7 1161.88     236 1125.55   295.7 1093.37   326.1 1085.73
   354.7 1070.28   402.5 1058.72     436 1035.14   478.7 1014.74   500.2 1009.31
   522.1  995.21   591.2  974.16   652.1  941.99   689.4  927.46   698.3  926.79
   704.1  927.48   771.7  931.88   790.3  939.13   842.5  940.32   863.3  954.99
   884.1  961.46   904.9  977.59   946.9  991.37  1021.3 1025.25  1059.1 1051.18
  1104.5  1064.7  1149.9 1084.66  1195.8 1114.64  1362.5 1202.63  1420.4 1238.64
#Mann= 5, -1 ,  0
       0     0.1       0   689.4   0.045       0   704.1     0.1       0
  800.39    0.06       0  954.76     0.1       0
Bank Sta=689.4,704.1
XS Rating Curve= 0 ,0
Exp/Cntr(USF)=0,0
Exp/Cntr=0.3,0.1

Type RM Length L Ch R = 1 ,97965   ,55.8,55.7,55.7
BEGIN DESCRIPTION:
Structure 22 XS 3
END DESCRIPTION:
XS GIS Cut Line= 3
1653601.52170295409130.5120094191653180.15689373409524.691992239
1652964.37733417 410374.21781728
#Sta/Elev= 30
       0  1166.5    67.4 1148.03    96.6 1134.71   143.5 1124.42   207.9 1091.26
   248.9 1074.31     325 1054.77   363.4 1032.67   443.9 1007.01   500.7  983.46
   585.1  938.05   616.4   933.2   770.4  925.93   786.9  921.49   791.4  920.76
   799.7  921.51   816.2  930.34   857.5  929.69     874  947.28   886.5  953.07
   944.1  975.41  1001.5   985.7  1018.4  998.44  1084.5 1017.45    1134 1042.46
  1175.9 1053.35  1212.4 1071.49  1241.3 1080.56    1427 1170.21  1453.5 1182.16
#Mann= 8, -1 ,  0
       0     0.1       0     577    0.07       0     617    0.06       0
   786.9   0.045       0   799.7    0.06       0     927     0.1       0
    1377    0.08       0    1427     0.1       0
Bank Sta=786.9,799.7
XS Rating Curve= 0 ,0
Exp/Cntr(USF)=0,0
Exp/Cntr=0.3,0.1

Type RM Length L Ch R = 1 ,97909   ,399.3,398.2,395.7
BEGIN DESCRIPTION:
Structure 22 XS 2
END DESCRIPTION:
XS GIS Cut Line= 4
 1653542.0548952409094.8319247681653125.78724093409504.303372438
1653113.89387937 409551.876818641652918.50293961410357.227300779
#Sta/Elev= 30
       0 1171.03    70.1 1148.87    95.9 1136.09   137.4 1125.18   254.3 1069.07
   300.1 1059.63   356.1 1034.81   487.3  987.34   580.6  941.17   625.4  934.94
   754.2  927.81   798.3  920.76   802.4  920.13   810.6  920.75   827.1  929.44
   868.2  928.09   901.2   947.5   923.1  956.09   946.4  962.81   975.3   963.7
  1008.2  979.66  1028.8  982.99  1086.4 1015.21  1127.5 1031.63  1148.1 1035.73
  1198.1 1057.35  1214.6 1067.89  1242.8  1075.2    1353 1132.34  1461.7 1177.62
#Mann= 10, -1 ,  0
       0     0.1       0     530    0.07       0  642.94    0.06       0
  772.94    0.05       0   798.3   0.045       0   810.6    0.05       0
  852.94    0.06       0  952.94     0.1       0 1192.94    0.08       0
 1452.94     0.1       0
Bank Sta=798.3,810.6
XS Rating Curve= 0 ,0
Exp/Cntr(USF)=0,0
Exp/Cntr=0.3,0.1

Type RM Length L Ch R = 1 ,97511   ,504,500,494.2
BEGIN DESCRIPTION:
Structure 22 XS 1
END DESCRIPTION:
XS GIS Cut Line= 6
1652910.47652726408975.1183714271652834.84610109409166.397188336
1652718.01398568409446.1650015121652689.28438434409532.831822917
1652681.25388859409607.7762268331652675.89267884 410358.14775759
#Sta/Elev= 30
       0  1099.1     126 1087.04   163.4 1089.03   233.9 1075.51   325.2 1050.47
     360 1027.54   390.4 1018.75   476.9  983.41   515.6  965.53   557.7  937.43
   587.2  925.84   607.9  920.44   720.3  918.46   728.3  917.11  737.66918.5488
   759.8  924.63   804.3  919.39   820.4  922.32   908.3  969.67   936.3  980.66
   952.3  982.76   972.3   995.9  1032.3 1018.08  1068.3 1042.24  1116.3 1054.91
  1144.3 1068.81  1168.3 1075.73  1364.3 1180.64  1408.3 1196.24    1426 1208.33
#Mann= 4, -1 ,  0
       0     0.1       0   720.3   0.045       0  737.66    0.06       0
  825.56     0.1       0
#XS Ineff= 2 , 0
                          782.17           952.5
Permanent Ineff=
       F       F
Bank Sta=720.3,737.66
XS Rating Curve= 0 ,0
Exp/Cntr(USF)=0,0
Exp/Cntr=0.3,0.1

Type RM Length L Ch R = 1 ,97011   ,493.3,495.2,489.7
XS GIS Cut Line= 6
1652029.89397085408938.4954131691652109.05326134409229.034530252
1652338.78541343409900.2323348371652356.81293643   409996.256421
1652363.02322584410201.5220865911652369.71054843410308.442148343
#Sta/Elev= 30
       0 1194.43    86.8 1158.51   138.7 1147.36     176 1133.38   248.2 1100.94
   306.3 1069.65   344.2 1053.92   388.5 1041.84   431.4 1016.69   617.3  955.86
   693.5  915.07   706.2  912.09  717.35915.1326   828.9  916.68   845.8  922.46
   879.8  921.87   908.1  931.82   985.5  973.35  1023.1  976.14  1051.6  987.53
  1063.8  993.99  1080.1 1009.07  1094.5 1011.93  1134.8 1038.47  1188.7 1054.06
  1208.7 1065.18  1228.7  1070.7  1336.8 1132.97  1352.8    1145  1420.8 1177.14
#Mann= 6, -1 ,  0
       0     0.1       0   693.5   0.045       0  717.35     0.1       0
  859.32    0.06       0  966.82    0.05       0 1070.57     0.1       0
Bank Sta=693.5,717.35
XS Rating Curve= 0 ,0
Exp/Cntr(USF)=0,0
Exp/Cntr=0.3,0.1

Type RM Length L Ch R = 1 ,96516   ,491.4,505,503.9
XS GIS Cut Line= 6
 1651614.5355496409058.7769967621651771.25570859 409555.02042684
1651795.27108051409652.7387353331651805.79107259409735.967243418
1651960.84883334410059.0991430881652111.90200892410425.762123674
#Sta/Elev= 30
       0 1183.76    41.1 1157.66    74.1 1149.87   127.5 1123.44   152.8 1106.69
   168.4 1102.28   224.5 1066.79   316.6 1033.61   358.5 1008.86   426.2  986.21
   457.8   968.7   499.8  956.17   575.3  924.25   620.9  911.43   745.2910.5825
   754.4  908.95   769.6  910.37   846.3  919.22   924.2  960.13   990.5  976.06
  1021.6  992.14  1047.5  997.15  1082.4  1012.3  1108.4 1030.53  1155.6 1044.75
  1208.2 1068.85    1351 1144.91  1368.2 1148.65  1424.2 1177.42    1460 1190.97
#Mann= 5, -1 ,  0
       0     0.1       0   745.2   0.045       0   769.6     0.1       0
  845.16    0.06       0  950.63     0.1       0
Bank Sta=745.2,769.6
XS Rating Curve= 0 ,0
Exp/Cntr(USF)=0,0
Exp/Cntr=0.3,0.1

Type RM Length L Ch R = 1 ,96011   ,498.3,500.5,501.6
XS GIS Cut Line= 6
1651552.24302326409060.4515340921651509.20931667409262.128624171
1651480.58503009 409462.954009921651461.36951734409647.658364922
1651417.47984134409817.0655064281651215.93398459410436.457640335
#Sta/Elev= 30
       0 1186.74    12.4 1183.04    40.1 1164.13    66.8 1152.72    98.7 1131.33
   143.5 1111.54   181.9    1089   192.4 1086.35   212.7 1069.71   257.2  1046.8
   289.6 1036.81     330 1013.93   370.4  995.79   394.6  989.02   426.8  972.45
     604  909.45   649.4  904.78     710905.6046   715.5  903.67   731.2  905.76
   740.3  911.45   769.3  914.17   886.8  912.48  1025.8  947.05  1072.1  966.22
    1091  970.67    1110  983.19  1240.5 1033.29    1354 1054.32  1421.2  1070.5
#Mann= 6, -1 ,  0
       0     0.1       0  709.82    0.07       0     710   0.045       0
   731.2    0.07       0  799.82    0.06       0  809.82     0.1       0
Bank Sta=710,731.2
XS Rating Curve= 0 ,0
Exp/Cntr(USF)=0,0
Exp/Cntr=0.3,0.1

Type RM Length L Ch R = 1 ,95510   ,232.1,229.8,227.2
BEGIN DESCRIPTION:
Structure 21.5 XS 4
END DESCRIPTION:
XS GIS Cut Line= 6
1651235.35979876 408926.70836325  1651092.404376409297.563592672
1651057.46284483409385.1500316711651023.48062934409466.142651841
1650993.35240875409535.0349025131650683.33137526410218.139507428
#Sta/Elev= 30
       0 1121.37    64.2 1102.72   190.6 1080.69   229.2 1062.64   254.9 1042.48
   294.7  1028.7   322.6 1006.69   338.1 1004.14   412.3  971.76   476.9  953.29
   544.3  919.45     584  904.79  699.46900.1707   709.2  898.85   715.3  900.21
   726.8  905.87     762  901.58   788.4  906.35   836.7  932.45   854.3  934.02
   937.6  963.27   968.4  980.03  1019.3  996.69  1043.1   999.3  1069.4 1022.08
  1112.3 1037.31  1223.1 1110.09  1303.4 1149.99  1341.7 1152.83  1404.9 1171.98
#Mann= 8, -1 ,  0
       0     0.1       0  599.59    0.06       0  699.46   0.045       0
   715.3    0.06       0  794.86     0.1       0  899.84    0.08       0
 1117.83     0.1       0 1226.22    0.08       0
Bank Sta=699.46,715.3
XS Rating Curve= 0 ,0
Exp/Cntr(USF)=0,0
Exp/Cntr=0.3,0.1

Type RM Length L Ch R = 1 ,95280   ,51,51,50.4
BEGIN DESCRIPTION:
Structure 21.5 XS 3
END DESCRIPTION:
XS GIS Cut Line= 3
1650750.75435343408762.4461201421650764.34676663409435.270573577
1650726.96763033410097.900717112
#Sta/Elev= 30
       0 1026.83    26.1 1014.25    49.7 1007.19    98.1 1002.27   138.1  989.77
   162.1  986.58   226.1  969.46   318.2   960.8   446.5  924.14   506.2  916.93
   706.3  902.94   727.5  898.42   734.3  897.93  740.14898.5421   750.4  902.83
   790.4  905.27   846.5  903.16   871.6   915.2   886.6  928.15   926.6  948.42
   978.7  959.63  1014.8  972.36  1038.8  974.35  1094.9  999.06  1118.9 1019.59
    1159  1034.1    1183 1053.18  1239.1 1086.05  1295.2 1116.95  1336.6 1135.16
#Mann= 11, -1 ,  0
       0     0.1       0     610    0.06       0  702.96     0.1       0
   727.5   0.045       0  740.14     0.1       0  802.96    0.06       0
  902.96     0.1       0 1002.96    0.05       0 1102.96    0.08       0
 1192.96     0.1       0 1292.96    0.08       0
Bank Sta=727.5,740.14
XS Rating Curve= 0 ,0
Exp/Cntr(USF)=0,0
Exp/Cntr=0.3,0.1

Type RM Length L Ch R = 1 ,95229   ,217.4,221,225
BEGIN DESCRIPTION:
Structure 21.5 XS 2
END DESCRIPTION:
XS GIS Cut Line= 6
1650720.17142373408762.4461201421650706.57901053409362.211352624
1650715.07426878409447.1639351281650711.67616548409521.922207732
1650706.57901053409606.8747902361650689.58849403410108.095027012
#Sta/Elev= 30
       0 1037.48    86.1 1020.71   186.1  990.95   242.2  985.74   296.8  976.27
   310.2   976.7   382.2  962.25   518.2  914.95   634.4  904.97   698.7  902.77
   708.8  898.08   714.7  897.29   722.7  898.09   750.7  904.91   850.9  903.68
   874.9  915.68   886.9  926.25   902.9  931.43   922.9  942.31   988.6  963.25
    1019  965.11    1039     978    1055  981.33    1071  990.69    1087  995.92
  1120.2 1020.99  1155.1 1034.47  1175.1 1051.67  1227.1 1083.06  1346.7 1147.57
#Mann= 8, -1 ,  0
       0     0.1       0   708.8   0.045       0   722.7     0.1       0
  800.13    0.06       0  905.24    0.08       0  995.24    0.05       0
 1095.24     0.1       0 1295.24    0.08       0
Bank Sta=708.8,722.7
XS Rating Curve= 0 ,0
Exp/Cntr(USF)=0,0
Exp/Cntr=0.3,0.1

Type RM Length L Ch R = 1 ,95008   ,498.8,497.5,485.2
BEGIN DESCRIPTION:
Structure 21.5 XS 1
END DESCRIPTION:
XS GIS Cut Line= 6
1650694.97505276408743.116866916  1650524.629921409376.207792342
1650403.80404717409609.3234678361650368.40451168409696.697308838
1650332.97151168 409893.932806761650316.60441843 410098.40779151
#Sta/Elev= 30
       0 1058.71    26.6 1054.43    51.2 1046.14    80.1 1045.61     105 1040.21
   299.4 1027.53   320.9  1019.2   353.1  1000.4   390.3   983.1     411  979.85
   431.6  971.24   555.8   930.2   614.2  900.75   696.5  898.07   709.5  896.66
  717.64898.1069   912.9  899.12   947.6  905.27   999.4  903.78    1049  914.72
    1078  929.57  1098.5  928.78  1151.2  944.63  1209.1  953.81  1239.8  962.27
    1272  966.23    1312  977.44  1332.2  980.56  1368.3  981.12  1418.3  991.74
#Mann= 8, -1 ,  0
       0     0.1       0   696.5   0.045       0  717.64     0.1       0
  755.67    0.05       0   870.7    0.06       0  978.28     0.1       0
 1082.56    0.08       0 1181.56     0.1       0
Bank Sta=696.5,717.64
XS Rating Curve= 0 ,0
Exp/Cntr(USF)=0,0
Exp/Cntr=0.3,0.1

Type RM Length L Ch R = 1 ,94511   ,513.2,500,484.5
XS GIS Cut Line= 6
1650078.60030125408645.8214578331650054.73551959408942.609906256
1650054.73551959409395.734984249 1649996.8534175409557.768452838
1650075.28009792409795.3808384981650242.70003867410104.617752835
#Sta/Elev= 30
       0 1180.98    14.8    1179    30.9 1180.73      51 1177.58    95.2 1160.43
   114.3 1155.64   151.7 1150.93   195.6 1128.68   299.7 1057.42   323.7 1049.93
   363.7 1028.81   394.4 1022.31   423.7 1012.19   451.7  996.99   483.7     991
   507.7  980.82   599.7  949.91  689.72894.8973   707.7  892.32   723.7  894.84
   962.9   893.3   984.3  894.14    1000  897.69  1020.5     895  1134.8  898.06
  1188.8  903.06  1291.9  905.55    1341  909.72  1400.6  933.61  1525.7  959.43
#Mann= 8, -1 ,  0
       0     0.1       0  689.72   0.045       0   723.7     0.1       0
  820.94    0.05       0  933.01     0.1       0 1067.61    0.05       0
 1137.61    0.07       0 1244.01     0.1       0
#XS Ineff= 2 , 0
                         1005.96          912.73
Permanent Ineff=
       F       F
Bank Sta=689.72,723.7
XS Rating Curve= 0 ,0
Exp/Cntr(USF)=0,0
Exp/Cntr=0.3,0.1

Type RM Length L Ch R = 1 ,94011   ,379.3,380.6,380
XS GIS Cut Line= 6
1649382.76223636409133.1075110341649561.91334251409394.651325002
1649659.48532584409416.554168344 1649855.8225316409556.583743915
1650040.02229442409795.0845792591650238.29256718410104.580679417
#Sta/Elev= 30
       0  983.33     9.2  979.41   112.6   947.7   161.9  924.84   171.8  923.79
   189.7  916.96   211.2  911.58   249.4  907.68   298.2  898.66     340  895.52
356.4282889.9774   364.6   887.5   370.9  887.96376.9282890.1785   389.2  891.33
   514.1  889.31   607.9   890.5   824.3  897.22     933  898.19   976.1  902.07
  1020.1   904.2  1105.2  904.57  1139.6  906.18  1157.4  910.31    1190  925.08
  1217.2  934.05    1237  938.02  1255.3  943.75  1270.6  945.58  1328.2  958.32
#Mann= 8, -1 ,  0
       0     0.1       0356.4282   0.045       0376.9282     0.1       0
  638.35    0.05       0  669.08     0.1       0  916.57    0.08       0
  946.57    0.07       0 1040.58     0.1       0
Bank Sta=356.4282,376.9282
XS Rating Curve= 0 ,0
Exp/Cntr(USF)=0,0
Exp/Cntr=0.3,0.1

Type RM Length L Ch R = 1 ,93630   ,110.8,119.4,133.9
XS GIS Cut Line= 6
  1649344.774927409159.1756856451649502.27701496409547.578892854
1649601.67153649409714.2558597271649646.01678456409752.484521854
1649673.54142129409796.8297699211649473.22323174410342.735065093
#Sta/Elev= 30
       0  975.01    40.3   961.2    96.4  945.95     118  935.78   148.2  928.59
     200   898.7     213  893.44   303.6  888.98   592.6  887.31  633.19884.4342
   644.9  884.18   653.4  884.44   671.7  887.96     762  895.78   771.6   902.6
   783.3  916.89   838.7  946.15   864.2  955.48   881.3  957.31   919.6  968.78
   936.7  970.12   952.4  975.55   996.3  993.18  1030.6  1013.1  1068.7 1024.27
  1094.3 1038.85  1119.9 1045.78  1234.9 1100.12  1256.2 1106.19  1305.4 1125.92
#Mann= 9, -1 ,  0
       0     0.1       0     220    0.08       0     260     0.1       0
     330    0.08       0  633.19   0.045       0   653.4    0.08       0
  663.19    0.07       0  681.73    0.06       0  793.93     0.1       0
Bank Sta=633.19,653.4
XS Rating Curve= 0 ,0
Exp/Cntr(USF)=0,0
Exp/Cntr=0.3,0.1

Type RM Length L Ch R = 1 ,93511   ,499.3,498.6,496.4
XS GIS Cut Line= 6
1649290.41519783409167.1914780891649337.01188943409297.152832344
1649393.32247233409433.7440945951649457.92831425409567.587658927
1649522.08304159409673.1258336751649261.96151459410376.988599166
#Sta/Elev= 30
       0  977.29    18.4  972.96    69.4  953.59   116.2  942.31   141.7  932.62
   219.6  891.91   232.6  889.31   449.6  888.33   477.7  886.24   524.5  887.65
599.9872884.9923   612.7  882.26624.3873884.9714   634.1  890.16   668.2  890.87
     698  911.76   727.9  923.74   753.5  938.38   779.1  942.45   817.4  953.94
   915.5  970.39   955.9  986.33   979.5   991.7   994.9 1000.36  1022.1 1010.97
    1069 1017.74    1133 1038.22  1172.4  1038.8  1253.4 1054.26  1308.3 1057.04
#Mann= 6, -1 ,  0
       0     0.1       0  218.06    0.08       0  544.43    0.06       0
599.9872   0.045       0624.3873    0.06       0  752.93     0.1       0
Bank Sta=599.9872,624.3873
XS Rating Curve= 0 ,0
Exp/Cntr(USF)=0,0
Exp/Cntr=0.3,0.1

Type RM Length L Ch R = 1 ,93012   ,511.9,506.7,496.4
XS GIS Cut Line= 6
1649037.93717257409173.5792062011649095.42444609409396.702502012
1649065.79130326409469.6328023371649004.41314517409820.950669259
1648980.79639451409915.1827642621648869.62404467410194.889553919
#Sta/Elev= 30
       0 1009.91    23.8   992.8    48.8  986.05    98.6  957.91   152.2  940.49
   176.9  929.65   201.5  916.06   213.9  905.44   232.9  899.89   260.5  884.03
   273.5   881.6   320.3  883.62352.9264879.9866   365.1  878.65372.7664879.9912
   405.9  881.59   422.1  886.49   474.8  885.06   564.1  893.34   653.3  897.21
   673.7  900.98   727.3  921.42   760.3  927.13   828.1   946.1     875  954.12
   905.2  962.55   926.3  972.09   987.4 1008.63  1026.7 1019.43  1064.1 1035.61
#Mann= 5, -1 ,  0
       0     0.1       0352.9264   0.045       0372.7664     0.1       0
   504.6    0.05       0  705.85     0.1       0
Bank Sta=352.9264,372.7664
XS Rating Curve= 0 ,0
Exp/Cntr(USF)=0,0
Exp/Cntr=0.3,0.1
